--- Twin Branch.prj (project) ---

Proj Title=Twin Branch
Current Plan=p01
Default Exp/Contr=0,0
English Units
Geom File=g01
Flow File=f01
Plan File=p01
BEGIN DESCRIPTION:
END DESCRIPTION:
DSS Export Rating Curves= 0
DSS Export Rating Curve Sorted= 0
DSS Export Volume Flow Curves= 0
DXF OffsetX= 0
DXF OffsetY= 0
DXF ScaleX= 0
DXF ScaleY= 0

--- Twin Branch.p01 (plan) ---

Plan Title=Floodplain
Program Version=4.00
Geom File=g01
Flow File=f01
K Sum by GR=0
Std Step Tol=0.01
Critical Tol=0.01
Num of Std Step Trials=20
Max Error Tol=0.3
Flow Tol Ratio=0.001
Split Flow NTrial=30
Split Flow Tol=0.02
Split Flow Ratio=0.02
Log Output Level=0
Friction Slope Method=1
Unsteady Friction Slope Method=2
Unsteady Bridges Friction Slope Method=1
Global Log Level=0
CheckData=False
Run HTab=0
Run UNet=0
Run PostProcess=0
UNET Theta=0
UNET Theta Warmup=0
UNET ZTol=0
UNET ZSATol=0
UNET MxIter=0
UNET MaxInSteps=0
UNET DtIC=0
UNET DtMin=0
UNET MaxCRTS=0
UNET WFStab=0
UNET SFStab=0
UNET WFX=0
UNET SFX=0
UNET DSS MLevel=0
UNET DZMax Abort=0
UNET Convert EG Bridges=0
UNET Use Existing IB Tables=0
UNET Froude Limit=0
UNET Froude Power=0
Write IC File=0
Echo Input=False
Echo Output=False
Write Detailed=0

--- Twin Branch.f01 (steady flow) ---

Flow Title=NFF Regression Equation
Program Version=4.00
Number of Profiles=1
Profile Names=P100yr
River Rch & RM=Twin Branch,Main      ,12458.6
615.2798
River Rch & RM=Twin Branch,Main      ,10433.3
648.9697
Boundary for River Rch & Prof#=Twin Branch,Main      ,1
Up Type=0
Dn Type=3
Dn Slope=0.017666

--- Twin Branch.g01 (geometry) ---

Geom Title=USGS 10m DEM
Program Version=4.00

River Reach=Twin Branch     ,Main
Reach XY= 30
     1773207.815      184512.232     1773149.748      184344.863
     1773081.721      183628.055     1773141.427      183397.282
     1773266.205      183271.161     1773522.471       183222.86
     1773877.353      183338.917     1773920.287      183305.375
     1774092.026      183344.284     1774251.689      183326.842
     1774376.468      183439.545     1774730.134      183553.203
      1774773.42      183471.441     1775459.315      183228.393
     1775740.984      181974.401     1775775.868      181728.198
     1775739.642      181468.578     1775834.903      181278.055
      1775965.72      180737.348      1776083.79      180657.516
     1776595.651      180018.863     1776731.834      179759.243
     1776848.563      179240.003     1776930.407        178742.9
     1776874.055      178434.308     1776221.129      177670.231
     1775520.273      176486.149     1775016.462      176100.409
     1774815.206      175796.512     1774700.457      175718.123

Type RM Length L Ch R = 1 ,12458.6 ,179.3,178,176.8
XS GIS Cut Line= 4
     1773607.739       184449.33       1773270.6      184483.044
     1773060.934      184513.759     1772813.588      184606.661
#Sta/Elev= 30
      10 1683.44    59.8 1653.04    89.7 1634.46   159.4 1589.08   189.3 1570.14
   219.2 1552.07   239.2 1540.54   249.1 1535.12   308.9 1505.43   318.9 1501.26
   369.1 1482.16   389.3 1473.71   399.4 1471.53   409.5 1472.01   411.9 1472.59
   419.5 1474.41   459.9 1487.78   490.2 1498.55   500.3 1502.58   520.5 1511.21
   530.5 1515.83   540.6  1521.1   550.7 1527.71   570.3 1542.81   580.1 1549.74
   736.7 1655.72   756.2 1670.02   785.6 1692.09   795.4 1698.92   814.9 1711.13
#Mann= 3 , 0 , 0
      10      .1       0   389.3    .045       0   411.9      .1       0
Bank Sta=389.3,411.9
XS Rating Curve= 0 ,0
Exp/Cntr=0.3,0.1

Type RM Length L Ch R = 1 ,12280.6 ,241.1,243.7,246.4
XS GIS Cut Line= 4
     1773570.279      184284.506     1773221.902      184310.728
     1773049.586      184344.442     1772817.334        184430.6
#Sta/Elev= 30
      10 1679.99    89.8 1624.52   109.8 1611.08   139.7  1591.8   179.7 1567.89
   229.6 1540.38   269.5  1520.6   339.4 1487.91   349.4 1484.21   359.1 1481.29
   414.9 1465.22   417.6 1464.49   427.4 1463.53   437.2 1464.65   439.9 1465.65
   446.9 1468.23   476.2 1480.94   505.4 1494.41   534.9 1509.03   554.7 1520.06
   594.3  1545.3   614.1 1559.16   633.9 1574.55   673.6 1607.48   683.5 1615.16
   693.4 1622.24   723.1 1642.56   742.9 1655.47   752.8  1661.5   772.7 1672.36
#Mann= 3 , 0 , 0
       0      .1       0   414.9    .045       0   439.9      .1       0
Bank Sta=414.9,439.9
XS Rating Curve= 0 ,0
Exp/Cntr=0.3,0.1

Type RM Length L Ch R = 1 ,12036.8 ,278,276.4,274.7
XS GIS Cut Line= 4
     1773522.768      184022.614     1773341.023      184063.938
     1773042.094       184093.46     1772717.788      184176.225
#Sta/Elev= 30
     9.8 1684.23    58.9 1640.53    78.5 1624.39    88.3 1616.97    98.1 1610.14
   107.9 1603.92     157 1574.57   226.4 1536.56   366.6 1463.92   376.6 1459.54
   386.6 1456.88   414.2  1453.2   426.7 1452.73  433.74 1454.43   436.7 1455.13
   466.7 1470.64   496.6 1484.21   516.3 1492.55     536 1499.55   565.5 1508.32
   575.4 1511.68   614.7 1527.47   624.6  1531.9   654.1 1548.26   683.6 1562.12
   713.2 1574.65   752.6 1589.49   772.2 1597.32   811.6 1614.68   821.5 1619.64
#Mann= 3 , 0 , 0
     9.8      .1       0   414.2    .045       0  433.74      .1       0
Bank Sta=414.2,433.74
XS Rating Curve= 0 ,0
Exp/Cntr=0.3,0.1

Type RM Length L Ch R = 1 ,11760.5 ,257.5,266.4,275.3
XS GIS Cut Line= 4
       1773516.8      183843.604     1773308.689      183784.088
     1772974.666      183834.987     1772708.701      183778.797
#Sta/Elev= 30
     9.8 1682.86    39.4 1663.48      59 1651.78    78.7 1641.46   127.9 1617.63
   147.6 1607.59   216.5 1569.27   315.8 1505.62   375.5 1468.09   385.4 1461.46
   405.3  1446.7   412.6 1443.91   415.2 1442.91   425.1 1442.74   437.6 1443.64
     445 1444.76   484.8 1452.88   604.7 1479.39   624.8 1485.36   634.9 1489.14
     655 1497.57   665.1 1502.35   685.2 1513.29   705.4 1525.62   715.4  1532.3
   735.6 1546.74   785.9 1586.75     796 1594.36     806 1601.34   826.2 1613.94
#Mann= 3 , 0 , 0
       0      .1       0   412.6    .045       0   437.6      .1       0
Bank Sta=412.6,437.6
XS Rating Curve= 0 ,0
Exp/Cntr=0.3,0.1

Type RM Length L Ch R = 1 ,11494.1 ,231,248,265.1
XS GIS Cut Line= 4
     1773536.565      183767.559     1773184.442      183569.021
      1772989.65      183535.307     1772794.858      183535.307
#Sta/Elev= 30
    10.1 1699.56    30.3 1689.25    50.5 1679.79    70.7 1670.92   121.3 1649.45
   141.5 1640.28   161.7 1630.39   171.8 1625.11   202.1 1608.51   262.8 1573.88
   303.2 1549.71   333.5 1531.12   404.2 1486.99   453.7 1454.47   473.4 1439.55
   480.7 1436.12   483.3 1434.89   493.2 1434.02   503.1 1436.15   542.6 1453.44
   562.4 1461.23   572.3 1464.78     592 1471.26   621.4 1479.48   631.1 1481.94
   650.6 1486.25   718.8 1499.26   757.8 1507.65   767.5 1509.36   796.7 1513.19
#Mann= 3 , 0 , 0
    10.1      .1       0   480.7    .045       0   503.1      .1       0
Bank Sta=480.7,503.1
XS Rating Curve= 0 ,0
Exp/Cntr=0.3,0.1

Type RM Length L Ch R = 1 ,11246.1 ,144.2,161.5,178.8
XS GIS Cut Line= 4
     1773557.319      183746.543     1773248.124      183385.467
     1773105.776       183243.12     1772875.709      183110.683
#Sta/Elev= 30
    10.1 1715.67    40.5 1704.79      91 1689.63   151.7 1669.26   192.2 1653.72
   212.4 1645.34   222.5 1640.58   232.6 1635.18   252.9 1623.16   293.3 1597.86
   364.1 1558.96   384.3 1547.25   404.6 1534.63     445 1508.53   465.3 1494.73
   505.6 1464.88   525.7 1448.53   535.8 1439.26   545.8    1432   553.5 1429.81
   555.9 1429.13     566 1428.86   578.5 1429.63   616.3 1434.16   686.5 1446.28
   755.3 1454.09   814.3 1465.54   853.7 1470.65     893    1475   942.1 1483.04
#Mann= 3 , 0 , 0
       0      .1       0   553.5    .045       0   578.5      .1       0
Bank Sta=553.5,578.5
XS Rating Curve= 0 ,0
Exp/Cntr=0.3,0.1

Type RM Length L Ch R = 1 ,11084.6 ,131.8,134.2,136.7
XS GIS Cut Line= 4
     1773589.009      183703.877     1773341.773      183329.278
      1773308.06      183119.502     1773188.188      183022.106
#Sta/Elev= 30
      10 1699.31    49.9 1685.83    89.8 1671.41   129.7 1655.58   149.6  1647.3
   169.6 1638.11   189.5 1626.93   229.4  1603.1   269.3 1578.78   279.3 1573.03
   299.2 1562.49   359.1 1533.51     389 1517.17   438.9 1488.43   458.5 1476.11
   487.5  1456.7   506.8 1443.34   526.1 1428.82  530.66 1427.54   535.8 1425.79
   548.2 1426.32     584 1430.51   603.4 1432.13     613 1432.54     671 1433.29
   699.9 1434.89   738.5    1439   786.8 1442.51   796.4  1443.8   815.8  1448.1
#Mann= 3 , 0 , 0
      10     .08       0  530.66    .045       0   548.2     .08       0
Bank Sta=530.66,548.2
XS Rating Curve= 0 ,0
Exp/Cntr=0.3,0.1

Type RM Length L Ch R = 1 ,10950.4 ,168.6,177,185.4
XS GIS Cut Line= 4
     1773596.501      183640.195     1773465.391      183295.564
     1773450.407      183078.296     1773439.169      182913.472
#Sta/Elev= 30
      10  1658.3    79.7 1621.45   129.6 1593.01   149.5 1581.35   159.5 1575.19
   199.3 1549.37   209.3 1543.15   219.2 1537.48   229.2 1532.37   259.1 1517.88
     299 1497.53   338.8  1478.3   368.7  1463.4   388.5 1452.39   408.3 1442.09
   428.1 1428.92   435.4 1425.86     438 1424.78   447.9  1423.5   460.4 1423.97
   507.3 1428.19   576.6 1433.74   586.5 1433.89   615.7 1433.01   625.4 1433.11
   635.1 1433.99   644.8 1437.29   664.3 1448.86   693.4 1464.73   751.7 1497.95
#Mann= 3 , 0 , 0
       0     .08       0   435.4    .045       0   460.4     .08       0
Bank Sta=435.4,460.4
XS Rating Curve= 0 ,0
Exp/Cntr=0.3,0.1

Type RM Length L Ch R = 1 ,10773.3 ,56,57.6,59.2
XS GIS Cut Line= 4
     1773652.801      183708.497     1773607.739      183359.246
     1773675.167      183078.296     1773633.982      182842.912
#Sta/Elev= 30
    10.1 1688.32    70.4 1651.88   130.8 1613.59   181.1  1580.1   261.6 1528.48
     332 1487.06   411.9 1443.51   421.9 1437.82   441.8 1424.83   449.2 1421.29
   451.8 1420.05   461.7 1419.45   474.2 1420.35   531.5 1425.55   541.4 1427.01
   551.4 1429.69   591.3 1443.24   601.2 1445.51   611.2 1446.18   631.1 1444.48
   641.1 1444.82     651 1446.89   690.9 1460.07   720.7 1470.71   740.6 1478.49
   750.6 1483.31   780.5 1498.99   800.4 1510.45   830.3 1529.02     880 1561.91
#Mann= 3 , 0 , 0
       0     .08       0   449.2    .045       0   474.2     .08       0
Bank Sta=449.2,474.2
XS Rating Curve= 0 ,0
Exp/Cntr=0.3,0.1

Type RM Length L Ch R = 1 ,10715.7 ,48.6,50.3,51.9
XS GIS Cut Line= 5
     1773686.405      183643.941     1773660.183      183359.246
     1773723.865       183149.47     1773746.341      182932.202
     1773753.833      182846.044
#Sta/Elev= 30
     9.9 1639.85      69 1601.54   118.3 1568.62   216.9 1505.44   256.3 1478.57
   266.2 1472.81   285.9 1463.31   335.7 1434.82   355.7  1421.5   363.1  1418.6
   365.6 1417.62   375.6 1417.52   388.1 1418.94   435.4 1423.49   445.3  1424.7
   455.3 1426.84   505.1 1444.23   515.1 1447.18     525 1448.77   534.9 1448.81
   554.8 1447.27   564.7  1447.5   574.6 1449.72   614.3 1464.78     664 1485.73
   673.9 1489.46   733.2  1508.7   742.8 1512.54   781.2 1529.83     810 1541.52
#Mann= 3 , 0 , 0
       0     .08       0   363.1    .045       0   388.1     .08       0
Bank Sta=363.1,388.1
XS Rating Curve= 0 ,0
Exp/Cntr=0.3,0.1

Type RM Length L Ch R = 1 ,10665.5 ,46.1,48.6,51.1
XS GIS Cut Line= 4
     1773716.373      183666.417     1773705.135      183359.246
     1773780.055      183153.216      1773839.99      182898.488
#Sta/Elev= 30
     9.9 1640.99    29.7 1632.56    39.7 1627.48    49.6 1621.66    99.2 1589.36
   128.9 1569.09   188.4 1530.01   218.1 1508.91   267.7 1468.91   277.6  1461.5
   287.5 1454.83   297.5 1449.12   317.3 1439.69   337.3 1431.01   367.2 1416.46
   377.1 1414.61   389.6 1415.75   456.9 1419.75   466.8 1421.66   476.8 1424.71
   536.7 1447.34   546.7 1448.95   566.9 1448.44   576.9 1448.73     587 1450.55
   597.1 1453.72   627.3 1465.57     738 1514.71   758.1  1522.5   788.3 1533.17
#Mann= 3 , 0 , 0
     9.9     .08       0   367.2    .045       0   389.6     .08       0
Bank Sta=367.2,389.6
XS Rating Curve= 0 ,0
Exp/Cntr=0.3,0.1

Type RM Length L Ch R = 1 ,10616.9 ,73.1,68.9,64.8
XS GIS Cut Line= 4
     1773757.579      183643.941     1773746.341      183366.738
     1773825.007      183198.168     1773854.974      183007.122
#Sta/Elev= 30
     9.9 1604.62    59.4 1585.99    69.4 1581.73    89.2 1571.23   148.6 1532.61
   168.4 1518.36   188.3 1502.11   237.8 1459.69   257.6 1444.82   267.5  1438.6
   287.2 1428.28     297 1423.92   316.6 1416.48   333.5 1412.27     346 1411.19
   358.5 1412.12   424.3 1413.26   434.1 1414.04   443.9 1415.94   463.5 1422.04
   511.8 1441.54   521.5 1444.59   531.1 1446.11   550.5  1447.4   560.1 1449.42
   579.5 1455.93   589.2 1460.47   608.5 1471.17   637.5  1488.4   656.8 1498.15
#Mann= 3 , 0 , 0
     9.9     .08       0   333.5    .045       0   358.5     .08       0
#XS Ineff= 2 , 0
                          406.82         1450.42
Permanent Ineff=
       F       F
Bank Sta=333.5,358.5
XS Rating Curve= 0 ,0
Exp/Cntr=0.3,0.1

Type RM Length L Ch R = 1 ,10548   ,115.3,114.6,113.1
XS GIS Cut Line= 4
     1773791.293      183670.163     1773819.344       183400.61
     1773890.433      183159.413     1773888.688      182958.424
#Sta/Elev= 30
      10  1591.3    40.1 1577.26   100.4 1550.29   150.6  1526.7   180.7 1510.44
   210.8 1491.79   240.9 1470.51     261 1454.83   291.1 1429.08   301.2 1421.37
   311.2 1415.33   321.3  1411.3   331.4 1408.07     339 1406.34   351.5 1405.35
     364  1406.1   431.9 1406.88     442 1407.22   452.1 1408.32   462.1  1410.7
   472.2 1414.01   542.6 1439.17   562.7 1444.51   572.7 1448.74   592.8 1460.89
     633 1482.73   683.3 1511.99   703.4 1525.52   713.4 1530.31   723.5    1534
#Mann= 3 , 0 , 0
      10     .08       0     339    .045       0     364     .08       0
#XS Ineff= 2 , 0
                          448.41         1495.94
Permanent Ineff=
       F       F
Bank Sta=339,364
XS Rating Curve= 0 ,0
Exp/Cntr=0.3,0.1

Type RM Length L Ch R = 1 ,10433.3 ,150.7,151.6,152.5
XS GIS Cut Line= 4
     1773976.281      183727.777     1773910.934      183413.259
     1773985.854      183158.531     1773951.593       182890.83
#Sta/Elev= 30
      10 1597.33   120.5 1522.27   170.7 1490.77   190.7 1480.21   210.8 1472.62
     251 1461.41     271 1453.66   311.2 1434.47   321.2 1429.14   350.7 1410.91
   360.6 1406.68   370.4 1404.69   390.1  1402.8   456.2  1402.4   468.7 1402.39
   481.2  1402.4   498.2 1402.48   508.1 1403.53   517.9  1406.3   567.1 1427.29
   626.7 1455.32   666.7 1475.71   706.7 1499.11   726.7 1512.88   756.7 1536.83
   786.7 1555.68   806.7 1565.82   816.7 1569.83   836.6 1576.09   856.6 1581.15
#Mann= 3 , 0 , 0
      10     .08       0   456.2    .045       0   481.2     .08       0
#XS Ineff= 2 , 0
                           512.1         1475.28
Permanent Ineff=
       F       F
Bank Sta=456.2,481.2
XS Rating Curve= 0 ,0
Exp/Cntr=0.3,0.1

Type RM Length L Ch R = 1 ,10281.7 ,214.3,219.9,221
XS GIS Cut Line= 4
     1774016.052      183718.861      1774046.02      183467.879
     1774135.924      183175.692     1774165.892      182984.646
#Sta/Elev= 30
    10.1 1596.09    30.3 1583.67    50.6 1570.16      91 1541.75   121.3 1521.46
   141.5 1506.88   171.9 1485.32   192.1 1472.35   202.2 1465.59   212.3 1458.29
   222.4 1451.46   232.5 1445.61   252.8 1435.01   302.1 1408.52   311.9  1404.2
   319.2 1402.88   321.8  1402.4   331.7 1402.38   344.2  1402.4   469.7 1402.45
   479.6 1403.23   489.4  1406.5   528.9 1428.89   548.6 1441.06   568.1 1452.71
   626.2 1486.58   655.2 1504.52   693.8 1529.15   703.5 1535.14   751.9 1564.16
#Mann= 3 , 0 , 0
    10.1     .08       0   319.2    .045       0   344.2     .08       0
Bank Sta=319.2,344.2
XS Rating Curve= 0 ,0
Exp/Cntr=0.3,0.1

Type RM Length L Ch R = 1 ,10061.8 ,133.6,131.4,132
XS GIS Cut Line= 3
     1774121.298      183760.665     1774276.315      183371.086
     1774424.366      182984.646
#Sta/Elev= 30
      10 1590.08    59.9  1556.2    99.8 1526.22   199.7 1454.05   219.6 1440.52
   239.6 1428.18   259.6 1416.78   279.5 1406.35   289.5 1403.18   299.5 1402.48
   329.4  1402.4   389.3 1402.37   459.7  1402.4  491.91 1402.67     500 1404.43
   510.1 1409.86   530.3 1423.37   540.4 1429.17   550.5 1433.84   560.6 1437.65
   570.7 1440.86   611.1 1452.37   621.2 1456.18   641.3 1465.26   671.6 1481.23
   681.7 1486.95   701.9 1499.46   782.6  1557.2   812.9 1576.94   833.1 1589.06
#Mann= 3 , 0 , 0
      10     .08       0   329.4    .045       0   459.7     .08       0
Bank Sta=329.4,459.7
XS Rating Curve= 0 ,0
Exp/Cntr=0.3,0.1

Type RM Length L Ch R = 1 ,9930.4  ,73.9,70.8,67.7
XS GIS Cut Line= 4
      1774252.05      183782.543     1774337.713      183601.609
     1774444.793      183249.027     1774547.983      183033.344
#Sta/Elev= 30
      10 1552.85    60.1 1517.86   150.1 1456.71   170.2 1444.27   200.2 1427.82
   230.1 1414.13     250 1406.53   259.9 1403.75   269.9 1402.46   309.7  1402.4
   369.5 1402.36   439.2  1402.4     499  1402.4   508.9 1402.93   518.9 1406.68
   528.8 1412.72   548.8 1426.04   558.7 1431.18   568.7 1435.06   618.5 1449.08
   628.4 1452.53   638.4 1456.97   648.4 1462.56   658.3 1468.97   698.2 1496.49
   708.1 1504.25     738 1529.16     758  1544.1   767.9 1552.13   807.8 1589.43
#Mann= 3 , 0 , 0
      10     .08       0   309.7    .045       0   439.2     .08       0
Bank Sta=309.7,439.2
XS Rating Curve= 0 ,0
Exp/Cntr=0.3,0.1

Type RM Length L Ch R = 1 ,9859.6  ,81.9,79.7,77.4
XS GIS Cut Line= 4
     1774322.047       183794.14     1774423.603      183618.955
     1774491.804       183254.25     1774575.937      183073.091
#Sta/Elev= 30
     9.6 1540.24    38.6 1519.81    77.1 1491.55    96.4 1479.15     135 1455.22
   154.3 1443.83   173.6 1433.32   192.9  1424.4   232.6 1410.55   242.6 1408.07
   262.7 1404.14   272.7 1402.88   282.7 1402.45   342.9  1402.4     403 1402.35
   453.2  1402.4   523.4  1402.5   533.4 1404.84   543.4 1410.49   563.5 1423.75
   573.5 1428.44   603.5 1435.57   613.5 1438.81   623.5 1443.11   633.4 1448.14
   643.4 1454.28   653.4 1461.77   693.4 1493.44   723.3 1518.01   773.3 1555.99
#Mann= 3 , 0 , 0
     9.6     .08       0   342.9    .045       0   453.2     .08       0
Bank Sta=342.9,453.2
XS Rating Curve= 0 ,0
Exp/Cntr=0.3,0.1

Type RM Length L Ch R = 1 ,9780    ,31.9,32.4,32.9
XS GIS Cut Line= 4
     1774405.774      183838.857     1774510.243      183657.082
     1774545.762      183308.156     1774611.665      183085.788
#Sta/Elev= 30
      10 1498.22    39.9 1480.39    69.9 1464.22   119.8 1442.03   159.7 1422.39
   169.7  1418.1   179.7 1415.31   189.7 1413.55   209.7 1412.11   259.8 1415.52
   299.8 1413.12   349.9 1414.72   357.5 1410.58     370 1402.34   382.5 1407.47
     390 1411.53   400.1 1415.05   410.1 1414.73   440.1 1409.29   460.2 1407.87
   480.2 1408.67   510.3 1412.71   530.3 1412.81   560.4  1414.5   620.9 1429.11
     631 1433.76   651.1 1446.72   691.5  1477.4   741.9 1513.61   792.3  1553.5
#Mann= 3 , 0 , 0
      10     .08       0   357.5    .045       0   382.5     .08       0
Bank Sta=357.5,382.5
XS Rating Curve= 0 ,0
Exp/Cntr=0.3,0.1

Type RM Length L Ch R = 1 ,9747.6  ,26.1,26.5,26.9
XS GIS Cut Line= 4
     1774448.992       183862.69     1774539.494      183659.171
     1774583.371       183293.53     1774649.566      183093.402
#Sta/Elev= 30
     9.7 1473.71    38.7 1458.24    58.1 1449.22   125.9 1425.45   145.3 1420.11
   154.9 1418.37     184 1414.29   193.7  1413.2   203.4  1412.9   213.1 1414.22
   222.7 1416.77   242.6 1420.45   262.5  1422.5   322.3 1422.23   352.1 1423.08
   362.1 1419.62     372 1410.03     382 1406.59  387.23 1409.89   401.9 1421.35
   411.8 1423.87   461.6 1422.96     581 1423.21   611.1 1424.21   621.1 1425.93
   631.1 1430.31   641.2 1436.82   711.5 1486.55   741.6 1509.09   801.8 1557.33
#Mann= 3 , 0 , 0
     9.7     .08       0     372    .045       0  387.23     .08       0
Bank Sta=372,387.23
XS Rating Curve= 0 ,0
Exp/Cntr=0.3,0.1

Type RM Length L Ch R = 1 ,9721.1  ,35.3,36.5,37.7
XS GIS Cut Line= 4
     1774490.655       183877.51     1774560.704       183677.35
     1774614.711      183285.173     1774705.315      183040.836
#Sta/Elev= 30
    10.1 1449.68    40.4  1435.7    50.5  1432.2    60.6 1429.98   131.3 1422.54
   191.9 1414.07     202 1414.24   231.9 1421.86   251.7 1423.73   261.5 1423.71
   291.2 1421.32   350.6 1422.13   360.5 1421.35   370.4 1411.41   373.9 1409.09
   380.3 1404.62  388.02 1409.09   400.1 1419.49     410 1422.57   469.4  1421.3
   538.7 1422.01   607.9  1423.9     618  1424.9     628 1427.92     638 1433.21
   678.1 1460.48   748.3 1513.65   798.4 1553.07   828.4 1574.57   868.5 1600.75
#Mann= 3 , 0 , 0
    10.1     .08       0   373.9    .045       0  388.02     .08       0
Bank Sta=373.9,388.02
XS Rating Curve= 0 ,0
Exp/Cntr=0.3,0.1

Type RM Length L Ch R = 1 ,9684.6  ,42.5,39.1,35.6
XS GIS Cut Line= 4
     1774572.767      183896.733     1774598.884      183627.726
     1774635.448      183426.624     1774692.906      183131.499
#Sta/Elev= 30
      10 1458.89      40 1448.58    50.1 1446.41    80.1  1442.1    90.1 1439.35
   130.1 1425.45   150.2 1421.28   190.2  1414.9   210.2  1413.7   220.2 1415.35
   240.2 1421.91   250.3  1421.9   289.7 1414.93   348.1 1412.11   357.9 1410.47
  371.86 1401.63   377.3 1397.99   387.1  1401.1   396.8 1408.75   406.5 1411.81
     426 1411.61   464.9 1407.82   524.8 1406.96   584.9 1409.59   594.9 1410.99
     605 1413.67     625 1422.23     645 1434.84   685.1 1463.89   775.3 1534.28
#Mann= 3 , 0 , 0
      10     .08       0  371.86    .045       0   387.1     .08       0
Bank Sta=371.86,387.1
XS Rating Curve= 0 ,0
Exp/Cntr=0.3,0.1

Type RM Length L Ch R = 1 ,9645.6  ,202.8,190.1,174.3
XS GIS Cut Line= 4
     1774725.733      183865.229     1774649.566      183626.572
     1774664.799      183370.143     1774725.733      183078.168
#Sta/Elev= 30
      10 1541.41    80.2 1496.92   100.2 1483.49   110.2 1475.51   120.2 1465.73
   140.3 1444.23   150.3 1435.86   170.4 1424.33   180.4 1420.32   190.4 1418.19
   230.5 1416.39   260.4 1411.29   299.9  1401.7   319.7 1395.95   336.8 1389.89
   339.4  1388.9   349.3 1388.65  355.31 1391.13   369.1 1395.35     379 1396.51
   497.5 1399.49   547.2 1402.15   557.1 1403.17   567.1 1405.61     577 1409.65
   596.9 1419.78   616.8 1432.63   656.5 1461.37   765.9 1545.42   805.7 1573.38
#Mann= 3 , 0 , 0
      10     .08       0   336.8    .045       0  355.31     .08       0
Bank Sta=336.8,355.31
XS Rating Curve= 0 ,0
Exp/Cntr=0.3,0.1

Type RM Length L Ch R = 1 ,9455.4  ,228.5,230.1,231.8
XS GIS Cut Line= 4
     1774806.457      183861.209     1774834.906      183591.027
     1774720.299      183250.612     1774765.251      183067.058
#Sta/Elev= 30
    10.1 1537.52    40.2 1520.37   120.7 1475.97   130.8 1470.68     161 1456.31
   191.2 1443.35   251.6 1419.34   271.7  1411.9   341.5 1391.63   351.5 1388.96
   381.4  1381.8   388.9  1380.5   391.4 1380.07   401.4 1379.67   413.9 1380.92
   441.3 1385.04   451.3 1386.05   461.2  1386.6   501.2 1386.37   541.1 1387.34
     551  1389.5     561 1394.06     571 1399.98     581 1406.47   610.9 1426.81
   650.8 1454.94   700.5 1492.05   770.1 1543.09     790 1556.66   819.8 1575.77
#Mann= 3 , 0 , 0
       0     .08       0   388.9    .045       0   413.9     .08       0
Bank Sta=388.9,413.9
XS Rating Curve= 0 ,0
Exp/Cntr=0.3,0.1

Type RM Length L Ch R = 1 ,9225.3  ,263.6,257.6,251.6
XS GIS Cut Line= 3
     1775119.653      183793.508     1775012.618      183398.244
     1774905.582       183002.98
#Sta/Elev= 30
      10 1566.68    59.9 1539.37    69.9 1533.28   109.9 1507.01   129.8 1494.86
   179.8 1465.46   209.7 1449.62   289.6 1411.18   349.6 1385.15   359.6  1382.3
     387 1376.75   399.5 1375.56     412 1376.16   479.4 1383.22   489.4 1384.68
   539.3 1396.25   559.3 1400.11   569.3 1402.89   579.3 1408.16   589.3 1415.02
   609.3 1430.23   629.2 1446.45   649.2 1463.62   689.2 1499.99   699.1 1508.25
   719.1 1523.45   749.1 1544.93     779 1564.92     799 1576.39     819 1586.74
#Mann= 3 , 0 , 0
       0     .08       0     387    .045       0     412     .08       0
Bank Sta=387,412
XS Rating Curve= 0 ,0
Exp/Cntr=0.3,0.1

Type RM Length L Ch R = 1 ,8967.7  ,216.9,203.9,190.7
XS GIS Cut Line= 3
     1775360.864      183673.909     1775304.674      183407.943
     1775065.884      182953.294
#Sta/Elev= 30
    10.1 1535.58    30.2 1524.21    50.3 1513.65    90.6 1493.37     141 1469.27
   221.5 1428.53   241.6 1419.67   261.8 1411.47     302 1393.01   322.2  1384.7
   332.3 1381.09   352.4  1375.5     360 1373.87   372.5 1372.39     385 1372.94
   463.2 1380.46   473.2 1381.59   483.3 1383.34   493.4 1386.04   523.6 1395.61
   543.7 1402.17   553.8 1405.86   563.9  1410.8   573.9 1417.11   624.3 1450.39
   664.5  1477.6   694.8 1497.14     735 1520.29   765.2  1536.2   785.4 1546.37
#Mann= 3 , 0 , 0
       0     .08       0     360    .045       0     385     .08       0
Bank Sta=360,385
XS Rating Curve= 0 ,0
Exp/Cntr=0.3,0.1

Type RM Length L Ch R = 1 ,8763.8  ,94.6,84.2,74.2
XS GIS Cut Line= 4
     1775631.116      183563.242     1775523.383      183298.806
     1775386.268      183191.073     1775121.831      183001.723
#Sta/Elev= 30
     9.8 1418.85    39.4 1413.02    78.8 1403.69   108.3 1397.38   137.8 1391.76
   147.7 1390.11   187.1  1384.4   206.8 1382.33   226.5 1380.78   265.8 1376.91
   285.5 1375.97   343.7 1371.53   369.9 1370.25   382.4 1369.79   392.1 1370.03
   394.9 1370.59   421.2 1375.75   430.9 1376.78   459.9  1378.2   499.3 1378.96
   519.1 1379.74   538.8 1381.01   548.6 1382.16   558.5 1384.33   627.5 1406.08
   637.3 1409.85   647.2 1414.74   666.9 1427.05   735.9 1472.01   785.2  1503.1
#Mann= 3 , 0 , 0
     9.8     .08       0   369.9    .045       0   394.9     .08       0
#XS Ineff= 2 , 0
          362.36 1385.64
Permanent Ineff=
       F       F
Bank Sta=369.9,394.9
XS Rating Curve= 0 ,0
Exp/Cntr=0.3,0.1

Type RM Length L Ch R = 1 ,8679.5  ,239.2,238.2,237.3
XS GIS Cut Line= 4
     1775731.717      183314.294     1775548.164       183186.93
      1775327.15      183119.502     1775147.342      182950.932
#Sta/Elev= 30
     9.7 1404.84    48.6  1402.8    77.7 1400.27   116.6 1396.18   145.7 1390.97
   155.4 1390.85   174.8 1392.92   184.6 1392.38   223.4 1384.87   263.6 1374.55
   281.2 1368.85   293.7 1366.49   303.8 1367.73   306.2 1368.56   323.9 1374.67
   333.9 1377.08     344 1378.38   374.1 1379.95   434.4 1381.27   444.4 1381.73
   454.5 1382.93   464.3 1385.43   523.5 1405.12   533.4 1408.58   543.2 1412.98
   553.1 1418.51   582.6 1436.11   622.1 1458.82   661.5 1482.62     701  1504.9
#Mann= 3 , 0 , 0
       0     .08       0   281.2    .045       0   306.2     .08       0
Bank Sta=281.2,306.2
XS Rating Curve= 0 ,0
Exp/Cntr=0.3,0.1

Type RM Length L Ch R = 1 ,8441.3  ,229.7,232.1,234.6
XS GIS Cut Line= 4
     1775915.271       183055.82     1775738.165      182990.073
     1775424.546       182905.98     1775115.195      182858.844
#Sta/Elev= 30
     9.9    1554    49.7 1527.71   129.3  1480.4   159.1 1461.83     179 1448.63
   188.9 1441.07   218.4 1420.43   238.1 1409.51     248 1405.19   257.8 1403.54
   287.3 1402.87   297.1 1401.23     307 1398.37   346.3 1383.05   402.7  1358.8
   405.4 1357.62   415.2 1355.55   425.1 1356.29   427.7 1357.08   493.9 1380.21
   533.8 1392.71   574.2 1404.24   584.3  1407.7   594.4 1412.13   624.7  1428.5
   654.9 1447.35   675.1 1459.09   715.5 1479.18   745.8 1495.87   826.5 1543.53
#Mann= 3 , 0 , 0
       0     .08       0   402.7    .045       0   427.7     .08       0
Bank Sta=402.7,427.7
XS Rating Curve= 0 ,0
Exp/Cntr=0.3,0.1

Type RM Length L Ch R = 1 ,8209.2  ,153.2,150.4,146
XS GIS Cut Line= 4
     1775960.223       182849.79     1775720.479      182759.887
     1775443.276      182658.745      1775177.31      182647.507
#Sta/Elev= 30
     9.8 1552.87    59.1 1525.07    68.9 1518.42    78.8 1510.83   118.2 1478.45
   147.7 1456.14   187.1 1430.68   216.7 1414.26   226.5 1409.13   246.2 1400.88
   305.2  1380.7   374.1  1358.4   391.1 1351.78   393.7 1350.75   403.6 1349.07
   413.4 1349.39   416.1 1349.96   423.3 1351.49   442.9 1357.45   501.9 1372.65
   511.8 1375.92   570.8 1399.72   580.7 1402.44   600.4 1406.55   610.3 1409.98
     699 1449.22     768 1482.68   787.7 1493.42   797.6 1499.73   817.3 1514.41
#Mann= 3 , 0 , 0
       0     .08       0   391.1    .045       0   416.1     .08       0
Bank Sta=391.1,416.1
XS Rating Curve= 0 ,0
Exp/Cntr=0.3,0.1

Type RM Length L Ch R = 1 ,8058.8  ,293.1,293.5,295.4
XS GIS Cut Line= 3
     1776018.614      182681.923     1775627.004      182563.746
     1775222.567      182484.986
#Sta/Elev= 30
      10 1482.99    49.9 1465.09    59.9 1459.74    99.8 1435.64   119.7 1425.58
   129.7  1421.5   139.7 1418.56   149.7 1416.82   199.5  1412.1   209.5  1409.5
   269.4 1384.73   299.3 1373.38   319.3 1367.39   379.1 1353.56   399.1 1346.18
   409.1 1343.48   419.1 1343.68   421.6 1344.36   449.3 1352.47   469.4 1356.36
   489.4 1361.68   549.7 1382.79   589.9 1395.21   630.1 1404.45   660.3 1408.21
   680.4 1411.53   720.6 1419.32   740.7 1423.84   770.8  1432.4   821.1 1450.74
#Mann= 3 , 0 , 0
      10     .08       0   399.1    .045       0   421.6     .08       0
Bank Sta=399.1,421.6
XS Rating Curve= 0 ,0
Exp/Cntr=0.3,0.1

Type RM Length L Ch R = 1 ,7765.3  ,220.6,219,217.3
XS GIS Cut Line= 4
     1776057.619      182389.033     1775871.169      182347.734
     1775536.925      182246.686     1775240.024      182170.663
#Sta/Elev= 30
    10.1 1482.99    40.2 1466.17    70.4  1448.6    90.5 1437.91   120.6 1424.07
   130.7 1419.85   160.8 1408.65   170.9 1403.97   250.8 1362.61   260.8 1358.46
   280.8 1354.27   330.6 1341.74   340.6 1340.47   370.5  1340.3   380.5 1339.32
   407.9 1334.75   420.4 1333.39   430.4 1334.56   432.9  1335.7   440.4 1339.09
   460.3 1350.08   569.8 1402.84   589.6 1412.93   609.4 1424.64   658.8 1455.02
   688.4 1471.32   718.1 1486.71   767.5 1510.57   807.1 1528.24   846.6 1545.12
#Mann= 3 , 0 , 0
       0     .08       0   407.9    .045       0   432.9     .08       0
Bank Sta=407.9,432.9
XS Rating Curve= 0 ,0
Exp/Cntr=0.3,0.1

Type RM Length L Ch R = 1 ,7546.3  ,224.9,221.4,218
XS GIS Cut Line= 4
     1776110.062      182141.798     1775926.509      182123.068
     1775626.829      182051.894     1775304.674      182006.942
#Sta/Elev= 30
     9.7 1473.78    29.1 1463.27    48.6  1451.2    87.4 1423.78   106.8 1411.21
   145.7 1389.65   165.1 1382.08   174.8 1376.63   204.4  1357.8   244.1    1334
   254.1 1330.43     264 1329.12   380.7 1327.91   393.2 1327.69   403.1 1327.88
   405.7 1328.81     413 1331.42   432.9 1344.58   442.8 1350.38   541.8  1404.5
   551.7 1408.73   561.5 1410.85   591.1 1411.75   600.9 1415.43   610.8 1423.35
   650.2 1463.25   699.5  1510.2   758.7 1563.87   788.2 1587.94   817.8 1608.22
#Mann= 3 , 0 , 0
     9.7     .08       0   380.7    .045       0   405.7     .08       0
#XS Ineff= 2 , 0
          325.75  1365.4
Permanent Ineff=
       F       F
Bank Sta=380.7,405.7
XS Rating Curve= 0 ,0
Exp/Cntr=0.3,0.1

Type RM Length L Ch R = 1 ,7324.9  ,155.9,154.5,153.6
XS GIS Cut Line= 4
     1776147.522      181984.466     1775907.779      181872.086
     1775664.289      181845.864     1775405.816      181845.864
#Sta/Elev= 30
     9.8 1412.72    68.6 1409.34    98.1 1406.46   107.9 1404.82   117.7 1401.02
   205.9 1355.94   215.7 1351.81   225.5 1348.69   294.2 1329.98     304 1327.76
   313.8 1326.41   343.1 1324.48   389.4 1322.48   401.9 1322.31   414.4 1322.41
   421.5 1322.59   431.3 1324.45   441.1 1329.84   450.9 1337.26   460.7 1343.88
   549.4 1398.08   559.4 1403.57   569.3 1406.67   599.1 1408.01   609.1 1411.14
     619 1417.72     629 1426.33   718.4 1508.68   738.3 1526.56   768.1 1552.47
#Mann= 3 , 0 , 0
     9.8     .08       0   389.4    .045       0   414.4     .08       0
#XS Ineff= 2 , 0
          351.63 1340.11
Permanent Ineff=
       F       F
Bank Sta=389.4,414.4
XS Rating Curve= 0 ,0
Exp/Cntr=0.3,0.1

Type RM Length L Ch R = 1 ,7170.3  ,325.1,335.8,345.3
XS GIS Cut Line= 3
      1776196.22      181711.008     1775795.322      181704.505
     1775385.949      181674.381
#Sta/Elev= 30
      10 1465.35    70.2 1425.63    90.2 1413.68   100.2 1409.97   130.3 1405.99
   140.3 1402.79   160.4 1391.38   210.5 1360.23   230.5 1350.28   260.6 1339.31
   320.8 1322.04   340.8 1318.64   368.4 1318.33   380.9 1318.31   393.4 1318.54
     421 1319.69     431 1321.83     461 1340.98   511.1 1370.06   541.1 1385.64
   571.1 1399.41   581.2 1402.58   591.2 1404.18   621.2 1406.65   631.2 1411.28
   641.2 1419.47   731.3 1508.18   741.3 1515.34   751.4  1520.2   811.4 1545.38
#Mann= 3 , 0 , 0
      10     .08       0   368.4    .045       0   393.4     .08       0
#XS Ineff= 2 , 0
          361.21 1338.29
Permanent Ineff=
       F       F
Bank Sta=368.4,393.4
XS Rating Curve= 0 ,0
Exp/Cntr=0.3,0.1

Type RM Length L Ch R = 1 ,6834.5  ,198.3,196.8,195.4
XS GIS Cut Line= 4
     1776176.922      181510.725     1775947.249      181456.088
     1775675.527      181355.139     1775417.054      181328.917
#Sta/Elev= 30
     9.8 1460.57    68.9 1425.48    88.5    1413    98.4  1408.2     118 1404.08
   127.9 1399.93   216.4 1347.72   236.1 1336.66   266.1 1320.93   276.1 1317.35
   286.1 1315.65   403.5 1310.44     416 1310.05     426 1310.58   428.5 1311.22
     436 1313.14     466 1325.61     506 1339.01   545.9 1357.44   595.9 1384.26
   615.9 1394.43   625.9 1399.01   635.9  1402.7   645.9 1405.03   655.9 1406.23
   705.8 1410.38   725.8 1413.16   735.8 1416.12   745.8 1420.16   785.8 1437.82
#Mann= 3 , 0 , 0
       0     .08       0   403.5    .045       0   428.5     .08       0
Bank Sta=403.5,428.5
XS Rating Curve= 0 ,0
Exp/Cntr=0.3,0.1

Type RM Length L Ch R = 1 ,6637.7  ,118,116.1,113.9
XS GIS Cut Line= 4
     1776203.712      181362.631     1775960.223      181246.505
     1775765.431      181186.569     1775454.514      181160.347
#Sta/Elev= 30
      10 1481.89    79.9  1432.7   109.9 1413.38   129.9 1401.54   209.8 1357.78
   279.5 1318.99   289.2 1315.01   298.9 1312.89   347.4 1308.44     364 1307.75
   376.5 1307.39   386.2 1308.36     389 1309.13   415.3 1317.04   473.6 1331.15
   483.6  1334.6   564.2 1370.38   624.5 1399.69   634.6 1404.08   644.7 1407.49
   654.7 1409.35   664.8 1409.95   705.1 1410.58   715.1 1411.78   725.2 1415.34
   735.3 1421.09   745.3 1428.33   765.5 1444.21   775.5 1451.04   785.6 1456.31
#Mann= 3 , 0 , 0
       0     .08       0     364    .045       0     389     .08       0
Bank Sta=364,389
XS Rating Curve= 0 ,0
Exp/Cntr=0.3,0.1

Type RM Length L Ch R = 1 ,6521.7  ,170.9,173.1,175.5
XS GIS Cut Line= 3
     1776248.151      181185.763     1775848.723       181093.67
     1775446.367      181017.901
#Sta/Elev= 30
      10 1508.29      50 1477.38     100 1440.15     130  1420.2     170  1395.2
     210 1369.15   269.9 1327.14   289.9 1313.97   299.9 1309.72   309.9 1308.14
   367.4 1305.83   379.9  1305.2   389.9 1306.24   392.4 1307.08   399.9 1309.61
   409.9 1313.97   419.9 1317.68   429.9 1320.08   459.8 1323.49   549.7  1331.1
   559.7 1332.32   569.7 1334.66   579.7 1338.15   649.6 1365.26   679.5  1376.3
   729.5 1393.67   749.4 1399.82   759.4 1401.78   769.4 1402.75   819.3 1404.35
#Mann= 3 , 0 , 0
      10     .08       0   367.4    .045       0   392.4     .08       0
#XS Ineff= 2 , 0
          328.98 1331.57
Permanent Ineff=
       F       F
Bank Sta=367.4,392.4
XS Rating Curve= 0 ,0
Exp/Cntr=0.3,0.1

Type RM Length L Ch R = 1 ,6348.6  ,277.8,295.9,314.1
XS GIS Cut Line= 4
     1776297.362      181070.444     1775986.445      180954.318
     1775772.923       180886.89     1775570.639      180845.684
#Sta/Elev= 30
    10.1 1503.89    50.3 1479.02    70.4 1464.82   110.6 1434.38   130.7 1421.09
   140.8 1415.41   150.9 1410.38   160.9 1406.29     181 1401.99   191.1 1396.81
   301.7 1322.54   321.8 1309.72   331.9 1305.96   341.6 1304.78   380.6 1302.66
   397.3 1300.67   409.8 1300.26   419.5 1302.85     439 1313.52   448.7 1316.21
   458.5 1316.39   526.6  1314.1   575.5 1313.21   585.3 1313.13   595.1  1314.2
     605 1318.14   644.3 1340.74   683.6  1360.9   722.9 1378.99   762.2 1395.36
#Mann= 3 , 0 , 0
    10.1     .08       0   397.3    .045       0   419.5     .08       0
Bank Sta=397.3,419.5
XS Rating Curve= 0 ,0
Exp/Cntr=0.3,0.1

Type RM Length L Ch R = 1 ,6052.6  ,182.5,175.6,168.7
XS GIS Cut Line= 4
     1776345.324      180970.892     1776147.522      180826.954
     1775990.191      180609.686     1775782.031      180364.613
#Sta/Elev= 30
     9.8  1494.5    29.4 1479.09    88.1 1427.28    97.9 1420.26   107.6 1416.63
     137 1418.62   146.8 1418.21   156.6 1414.97   274.4 1338.03   324.1 1307.19
     334 1302.36     344 1299.85   393.7 1294.49   420.9 1287.22   433.4 1286.59
   445.9 1291.26     493 1317.41   583.2 1372.73   623.4 1395.92   633.5 1399.68
   643.5 1401.18   663.6 1400.91   673.7 1401.81   683.7 1405.53   693.7 1413.34
   703.8 1424.12   723.9 1449.84   733.9 1460.99   794.2 1513.65   834.4  1547.5
#Mann= 3 , 0 , 0
       0      .1       0   420.9    .045       0   445.9      .1       0
Bank Sta=420.9,445.9
XS Rating Curve= 0 ,0
Exp/Cntr=0.3,0.1

Type RM Length L Ch R = 1 ,5877.1  ,206.5,204.7,202.8
XS GIS Cut Line= 4
     1776443.456      180819.462      1776214.95      180602.194
     1776068.857      180478.577     1775855.335      180332.483
#Sta/Elev= 30
     9.9 1413.34    49.3 1415.89    59.1 1415.83    78.8 1414.66    88.7  1412.4
    98.5  1408.9   108.4 1404.11   128.1 1391.86   157.7 1370.97   167.5 1365.19
   216.8 1339.01   226.6 1334.14   246.3 1325.42   305.5 1300.58   315.3 1296.87
   325.4 1294.51   365.7 1289.54   383.4 1286.56   385.8 1286.18   395.9  1286.1
     406 1289.34   426.1 1303.99   436.2 1310.62   516.6 1361.09   576.3 1397.15
   606.2 1416.49   626.1 1430.27   685.8 1473.39   725.6 1503.39   765.4 1534.37
#Mann= 3 , 0 , 0
     9.9      .1       0   383.4    .045       0     406      .1       0
Bank Sta=383.4,406
XS Rating Curve= 0 ,0
Exp/Cntr=0.3,0.1

Type RM Length L Ch R = 1 ,5672.4  ,212.2,213.5,214.8
XS GIS Cut Line= 4
     1776604.018      180646.671     1776442.308      180509.902
      1776196.22      180328.737     1775978.687      180117.784
#Sta/Elev= 30
    10.1  1349.2    40.3 1339.88    80.7 1325.21     121 1311.95   151.3 1304.75
   211.8 1299.28   270.9 1296.28   290.7 1294.13   330.1 1291.79   396.4 1281.31
   408.9 1279.91   418.8 1280.76   421.4 1281.96   428.7 1285.34   458.2 1310.53
   567.9 1393.33     578  1399.7   598.2 1410.12   618.4 1424.49   628.5 1433.56
   648.7 1455.32   668.9 1479.88   689.1 1507.56   699.2 1519.33   709.3 1527.42
   719.4 1533.63   739.6 1543.48     780 1560.58   800.2 1570.23   820.4 1578.12
#Mann= 3 , 0 , 0
       0      .1       0   396.4    .045       0   421.4      .1       0
Bank Sta=396.4,421.4
XS Rating Curve= 0 ,0
Exp/Cntr=0.3,0.1

Type RM Length L Ch R = 1 ,5458.9  ,225.1,220.7,216.4
XS GIS Cut Line= 4
     1776713.167      180512.291      1776514.63      180306.261
     1776316.092      180145.183     1776098.825      180017.819
#Sta/Elev= 30
     9.9 1414.87    19.7 1413.06    29.6 1408.47    59.2 1387.85    88.8 1368.63
   108.5 1356.74   197.3 1310.85   217.1 1301.92   226.9 1298.67   236.8 1296.38
   246.7 1295.06   325.5 1285.61   374.6 1281.64   384.5 1280.12   401.5 1274.87
   404.1 1274.01     414 1273.05   423.8 1275.09   426.5 1276.52   522.1 1330.84
   561.9  1351.3   602.2 1369.95   632.4  1381.5   682.8 1397.26   692.9 1399.33
   733.2 1403.37   753.3  1408.1   763.4 1412.06   773.5 1417.35   793.6 1430.65
#Mann= 3 , 0 , 0
       0      .1       0   401.5    .045       0   426.5      .1       0
Bank Sta=401.5,426.5
XS Rating Curve= 0 ,0
Exp/Cntr=0.3,0.1

Type RM Length L Ch R = 1 ,5238.2  ,243.7,242.2,240.7
XS GIS Cut Line= 4
     1776883.173      180324.266     1776713.167      180148.929
     1776447.202      179995.343     1776224.297      179837.807
#Sta/Elev= 30
     9.8 1411.35    19.5 1404.16    29.3  1401.1    48.8 1402.99    58.6 1402.71
    68.4 1399.85   107.5 1378.84   185.6 1331.16   205.1  1320.5   244.2  1302.6
   293.8 1283.64   303.7 1280.46   313.6 1279.11   392.8 1276.63   402.7 1275.27
     420 1270.72   432.5  1269.6     445 1273.71   472.1 1288.67   591.8 1348.47
   632.2    1368   682.8 1390.44     703  1396.9   713.1 1398.76   723.2 1399.44
   753.5 1398.65   773.8  1400.9   783.9 1405.26   804.1 1416.53   824.3 1424.99
#Mann= 3 , 0 , 0
       0      .1       0     420    .045       0     445      .1       0
Bank Sta=420,445
XS Rating Curve= 0 ,0
Exp/Cntr=0.3,0.1

Type RM Length L Ch R = 1 ,4995.9  ,230.1,224.6,219
XS GIS Cut Line= 4
     1776997.863      180074.009     1776788.087       179905.44
     1776544.598      179781.822     1776312.346      179714.394
#Sta/Elev= 30
      10 1422.96    19.9 1414.15    29.9  1406.4    39.9 1401.65    49.8 1400.58
    69.8 1401.74    79.7 1399.13    89.7 1393.12   149.5 1349.08   179.4 1328.41
   229.2 1297.66   259.1 1280.98   269.1 1277.79   279.2 1276.45   360.1 1270.59
     378 1268.51   390.5 1267.12     403 1267.81   410.7 1269.41     441 1278.52
   461.3 1285.65   481.5 1294.33   501.7 1304.79     522 1316.92   572.4 1351.44
   592.6 1367.86   622.8 1395.69   632.9 1402.82   743.7  1457.1     784 1478.48
#Mann= 3 , 0 , 0
       0      .1       0     378    .045       0     403      .1       0
Bank Sta=378,403
XS Rating Curve= 0 ,0
Exp/Cntr=0.3,0.1

Type RM Length L Ch R = 1 ,4771.4  ,323.4,319.1,314.7
XS GIS Cut Line= 4
     1777137.853      179819.787     1776979.133      179703.156
     1776638.248      179609.506     1776348.061      179602.957
#Sta/Elev= 30
     9.8 1357.31    39.4 1353.13    78.8 1348.75    88.6 1347.07    98.5 1344.66
     128 1334.77   187.1 1319.04   227.3 1306.47   287.9 1283.04     298 1280.25
   358.6 1269.66   368.7 1268.24     399 1265.73   416.8 1263.43   429.3    1262
   439.4 1263.39   441.8 1264.53   449.5 1268.18   459.6 1273.79   469.7 1278.51
   560.5 1316.65   580.5 1325.64   600.5 1335.57   630.6  1352.3   660.6 1370.65
   700.6 1398.39   710.6 1407.05   730.6 1425.66   740.7 1433.35   840.7    1499
#Mann= 3 , 0 , 0
       0      .1       0   416.8    .045       0   441.8      .1       0
Bank Sta=416.8,441.8
XS Rating Curve= 0 ,0
Exp/Cntr=0.3,0.1

Type RM Length L Ch R = 1 ,4452.3  ,168.2,167.4,166.6
XS GIS Cut Line= 4
     1777230.959      179409.133     1777035.323      179354.779
     1776698.184      179317.319     1776423.427      179271.789
#Sta/Elev= 30
     9.7 1399.62    38.7 1395.68    48.3 1393.38      58 1389.77    77.4 1379.36
   106.4 1360.58     116 1355.98     174 1337.74     223 1314.31   252.9 1301.64
   302.8 1285.06   362.7 1262.65   372.7 1260.42   400.1 1258.03   412.6 1257.02
   422.5 1257.56   425.1 1258.82   432.5 1262.41   452.5 1278.56   462.4 1285.58
   621.8 1393.17   631.8  1397.4   641.7 1399.04   661.6 1400.38   671.6 1404.63
   691.5 1422.17   711.4 1437.53   761.1 1479.53   790.9 1508.99   820.8 1534.68
#Mann= 3 , 0 , 0
       0      .1       0   400.1    .045       0   425.1      .1       0
Bank Sta=400.1,425.1
XS Rating Curve= 0 ,0
Exp/Cntr=0.3,0.1

Type RM Length L Ch R = 1 ,4284.9  ,201.4,200.9,200.5
XS GIS Cut Line= 4
     1777245.099      179238.653     1776952.911      179174.971
     1776724.405      179156.241     1776473.424      179152.495
#Sta/Elev= 30
      10 1426.13    29.9 1410.48    39.9 1405.08    49.8  1402.7    79.7 1402.56
    89.7 1400.62    99.7 1396.01   129.6 1377.53   149.5 1363.57   179.4 1340.02
   199.4 1320.63   209.3 1312.85   229.3 1302.35     299 1274.88   338.9 1261.41
   348.9 1259.44   378.8 1256.75   396.2 1254.09   408.7 1253.53   418.7 1256.49
   438.6 1268.61   498.4 1301.14   538.4 1324.19   588.6 1356.45   628.7 1385.19
   638.8 1388.12     709 1398.37   719.1 1402.77   749.2 1428.28   779.3 1457.81
#Mann= 3 , 0 , 0
      10      .1       0   396.2    .045       0   418.7      .1       0
Bank Sta=396.2,418.7
XS Rating Curve= 0 ,0
Exp/Cntr=0.3,0.1

Type RM Length L Ch R = 1 ,4084    ,438.9,433.1,427.3
XS GIS Cut Line= 4
     1777281.547      179004.964     1777072.783      178980.179
     1776784.341      178961.449      1776472.07       178880.43
#Sta/Elev= 30
      10 1405.38      40 1395.61    50.1 1390.93    90.1 1366.47   110.1  1355.5
   150.2 1336.88   220.2 1306.98   250.1 1290.43   299.9 1259.41   309.9 1255.77
   319.9 1254.33   397.1  1249.5   409.6 1248.86   422.1 1251.78   439.5 1259.95
   449.4  1263.6   549.7 1297.92   569.8 1306.27   579.9 1311.78     590 1319.29
   600.1 1329.55   640.4 1373.51   660.6 1393.92   670.7 1400.52   690.8 1408.39
   700.9 1415.44   741.2 1450.32   771.5 1480.71   791.6 1495.85   821.9 1515.16
#Mann= 3 , 0 , 0
       0      .1       0   397.1    .045       0   422.1      .1       0
Bank Sta=397.1,422.1
XS Rating Curve= 0 ,0
Exp/Cntr=0.3,0.1

Type RM Length L Ch R = 1 ,3650.9  ,200.9,187.6,174.3
XS GIS Cut Line= 4
     1777301.288      178523.168     1777096.267      178521.164
     1776784.341      178564.374      1776497.06      178645.648
#Sta/Elev= 30
     9.8 1332.12    58.6 1324.09    87.9 1317.99   185.5 1294.35   224.7 1283.96
   254.2 1275.06   273.9 1267.79   283.8 1262.73   303.4 1250.31   313.3  1244.9
   323.1 1242.44   362.5 1243.12   379.5 1238.62     392  1236.3   404.5 1237.86
   421.5  1242.9   431.4 1247.33   451.1 1258.69   569.7 1330.64   589.6 1343.98
   659.3 1392.72   669.2 1398.89   689.1 1409.15     709 1420.26   748.8 1444.89
   768.7 1454.98   788.6 1463.32   798.6 1467.02   808.5 1469.72   818.5 1471.05
#Mann= 3 , 0 , 0
       0      .1       0   379.5    .045       0   404.5      .1       0
Bank Sta=379.5,404.5
XS Rating Curve= 0 ,0
Exp/Cntr=0.3,0.1

Type RM Length L Ch R = 1 ,3463.3  ,189.7,184.6,179.4
XS GIS Cut Line= 4
     1777173.925      178253.457     1776919.197      178317.138
     1776761.865      178429.518     1776507.138      178556.882
#Sta/Elev= 30
    10.1  1406.3    20.2 1404.07    30.3 1399.67    50.5 1386.35    70.7 1371.27
    80.8 1364.28   161.6 1314.23   191.9 1294.92     202  1288.7   212.1 1283.31
   262.6 1261.07   291.6 1245.74   301.2 1241.87   310.9 1240.68   330.2 1240.66
   339.9 1239.47   346.7 1237.27   359.2 1234.28   368.9 1234.69   371.7 1235.66
   378.6 1238.05   397.9 1248.73   514.8 1322.28   544.3 1340.17   622.9 1384.03
   642.5    1394   652.3 1398.07   662.1  1401.1   691.6  1406.7   740.7 1414.67
#Mann= 3 , 0 , 0
       0      .1       0   346.7    .045       0   371.7      .1       0
Bank Sta=346.7,371.7
XS Rating Curve= 0 ,0
Exp/Cntr=0.3,0.1

Type RM Length L Ch R = 1 ,3278.8  ,248.5,248,247.6
XS GIS Cut Line= 4
     1776990.371      178017.459     1776803.071      178144.823
     1776634.502      178320.884      1776400.64      178504.133
#Sta/Elev= 30
     9.8 1361.84    49.2 1345.38    68.9 1337.98   118.2 1321.11   157.6  1308.4
   187.1 1299.76   206.8 1294.66   226.5 1289.92   265.5  1282.8   275.3 1279.85
     285 1275.27   294.8 1268.91   333.8 1241.42   343.5 1235.32   350.5 1232.38
   353.3  1231.2     363 1230.42   372.8 1232.33   375.5  1233.6   382.5 1236.89
   470.2 1286.46   509.9 1307.03   569.3 1330.81   608.9 1345.74   628.7 1352.21
   638.6 1354.69   648.5 1355.61   678.2  1354.3   688.1 1355.48   767.4 1369.52
#Mann= 3 , 0 , 0
       0      .1       0   350.5    .045       0   375.5      .1       0
Bank Sta=350.5,375.5
XS Rating Curve= 0 ,0
Exp/Cntr=0.3,0.1

Type RM Length L Ch R = 1 ,3030.7  ,165.5,171.6,177.7
XS GIS Cut Line= 4
     1776863.007      177822.667     1776612.026      177983.745
     1776465.932      178141.077     1776241.172      178272.186
#Sta/Elev= 30
     9.9 1405.86    39.8    1408    49.7  1406.1    59.6 1401.18   149.1 1336.62
   178.9 1315.84   238.6 1277.72   248.5 1271.76   258.5 1266.72   278.3 1258.76
   298.2 1252.74   317.7 1249.01   356.8 1244.38   366.5 1242.01   376.3 1238.38
   395.8 1232.76   412.6 1226.78   415.3 1225.77   425.1 1225.33   434.9 1228.82
   454.4 1237.57   464.1 1242.54   522.9 1279.41     583 1313.96     623 1333.45
   683.1 1365.28   703.1 1373.78   723.1 1380.16   743.1 1387.74   773.1 1402.56
#Mann= 3 , 0 , 0
     9.9      .1       0   412.6    .045       0   434.9      .1       0
Bank Sta=412.6,434.9
XS Rating Curve= 0 ,0
Exp/Cntr=0.3,0.1

Type RM Length L Ch R = 1 ,2859.1  ,207.6,207.2,206.9
XS GIS Cut Line= 3
      1776761.44      177704.762     1776423.909      177936.632
     1776086.379      178168.502
#Sta/Elev= 30
      10 1395.48      30 1384.45      40 1380.27    59.9 1374.02    69.9  1369.8
    79.9  1364.5   119.9 1336.28   149.8 1319.35   159.8  1314.6   189.8 1303.24
   229.7 1285.47   299.6 1251.45   309.6 1247.26   329.6 1240.67   379.5  1228.3
     397  1222.3   409.5 1219.71   419.5  1220.7     422 1221.63   429.5 1224.41
   449.5 1233.82   559.3 1287.34   579.3 1298.65   609.3 1318.54   629.2 1330.42
   719.1 1377.24   739.1 1385.88   759.1 1393.22     779 1399.28     819 1409.49
#Mann= 3 , 0 , 0
       0      .1       0     397    .045       0     422      .1       0
Bank Sta=397,422
XS Rating Curve= 0 ,0
Exp/Cntr=0.3,0.1

Type RM Length L Ch R = 1 ,2651.9  ,194.8,196.5,198.3
XS GIS Cut Line= 4
      1776664.47      177601.654      1776402.25       177699.05
     1776199.966      177841.397     1775997.683      177968.761
#Sta/Elev= 30
      10  1399.3      50 1401.36    59.9 1400.39    69.9 1398.67    79.9 1396.18
    99.9 1388.65   109.9 1384.12   119.9 1378.78   129.9 1372.56   189.8 1333.57
   259.7 1292.12   319.3 1258.39   378.7  1226.8   395.8 1217.16   398.5 1215.76
   408.3 1213.42   418.2  1214.2   420.8 1214.94   447.9  1222.9   477.6 1229.05
   487.5 1232.35   497.4 1236.46   517.2 1246.83   566.9 1278.37   586.8 1289.92
   606.8 1299.43   676.5 1328.01   686.4 1332.55   696.4 1338.03   766.1 1383.42
#Mann= 3 , 0 , 0
       0      .1       0   395.8    .045       0   420.8      .1       0
Bank Sta=395.8,420.8
XS Rating Curve= 0 ,0
Exp/Cntr=0.3,0.1
